--- CABINCK.prj (project) ---

Proj Title=CABINCK
Current Plan=p01
Default Exp/Contr=0,0
English Units
Geom File=g01
Flow File=f01
Plan File=p01
BEGIN DESCRIPTION:
END DESCRIPTION:
DSS Export Rating Curves= 0
DSS Export Rating Curve Sorted= 0
DSS Export Volume Flow Curves= 0
DXF OffsetX= 0
DXF OffsetY= 0
DXF ScaleX= 0
DXF ScaleY= 0

--- CABINCK.p01 (plan) ---

Plan Title=Floodplain
Program Version=4.00
Geom File=g01
Flow File=f01
K Sum by GR=0
Std Step Tol=0.01
Critical Tol=0.01
Num of Std Step Trials=20
Max Error Tol=0.3
Flow Tol Ratio=0.001
Split Flow NTrial=30
Split Flow Tol=0.02
Split Flow Ratio=0.02
Log Output Level=0
Friction Slope Method=1
Unsteady Friction Slope Method=2
Unsteady Bridges Friction Slope Method=1
Global Log Level=0
CheckData=False
Run HTab=0
Run UNet=0
Run PostProcess=0
UNET Theta=0
UNET Theta Warmup=0
UNET ZTol=0
UNET ZSATol=0
UNET MxIter=0
UNET MaxInSteps=0
UNET DtIC=0
UNET DtMin=0
UNET MaxCRTS=0
UNET WFStab=0
UNET SFStab=0
UNET WFX=0
UNET SFX=0
UNET DSS MLevel=0
UNET DZMax Abort=0
UNET Convert EG Bridges=0
UNET Use Existing IB Tables=0
UNET Froude Limit=0
UNET Froude Power=0
Write IC File=0
Echo Input=False
Echo Output=False
Write Detailed=0

--- CABINCK.f01 (steady flow) ---

Flow Title=NFF Regression Equation
Program Version=4.10
Number of Profiles= 1
Profile Names=P100yr
River Rch & RM=CABINCK,Main            ,17881.3
647.1305
River Rch & RM=CABINCK,Main            ,17077.1
1062.478
River Rch & RM=CABINCK,Main            ,15783.3
1104.462
River Rch & RM=CABINCK,Main            ,13101.2
 1208.91
River Rch & RM=CABINCK,Main            ,9845.2
1339.535
River Rch & RM=CABINCK,Main            ,7749.6
1488.198
River Rch & RM=CABINCK,Main            ,5043.4
1640.682
River Rch & RM=CABINCK,Main            ,449.4
1809.755
Boundary for River Rch & Prof#=CABINCK,Main            , 1
Up Type= 0
Dn Type= 3
Dn Slope=0.018
DSS Import GetInterval= 0
DSS Import GetPeak= 0
DSS Import FillOption= 0

--- CABINCK.g01 (geometry) ---

Geom Title=USGS 10m DEM
Program Version=4.10

River Reach=CABINCK         ,Main
Reach XY= 30
     1858619.513      361874.114     1858387.723      361894.142
      1858159.48      362154.814     1857564.268      363528.086
     1857516.603      364088.073     1857231.522      364359.105
     1857185.171      364636.688     1856654.026      365416.892
     1856555.048      366101.565       1856088.8      366295.106
     1855639.937      366957.108      1855580.12      367282.953
      1855254.68       367660.82     1855142.238      368077.186
     1854820.027      368596.238     1854009.023      369575.032
     1853783.103      370135.969     1853226.685       370646.38
     1853062.574      370732.322     1852939.802      370679.877
     1852497.135      371144.603     1851685.645      371496.593
     1850622.955      370774.508     1850269.979      370733.615
     1849948.657       370911.31     1849464.276      370549.011
     1848933.234       370647.17     1848428.601      370333.724
     1848172.321      370369.461     1847365.502      370869.213

Type RM Length L Ch R = 1 ,17881.3 ,228.8,216.3,203.7
XS GIS Cut Line= 3
     1858594.523      361693.693     1858600.355      361945.679
     1858629.234      362045.552
#Sta/Elev= 27
       0 1645.73    38.8 1614.19    48.5 1606.48    58.2 1600.12    67.9 1597.22
     126 1592.26   135.7 1590.41   145.4 1586.22   155.1 1580.72   164.8  1575.4
   174.5  1571.3   180.91570.375   184.2  1569.9   193.9 1569.84   203.6  1569.7
   213.3 1570.18     223 1571.37   242.4 1574.46     271 1579.39   280.4  1580.9
   289.9  1582.1   299.3 1582.93   318.2 1584.28   327.7 1585.13   337.1 1586.32
   346.6 1589.24     356    1594
#Mann= 3 , 0 , 0
       0      .1       0   180.9    .045       0   193.9     .08       0
Bank Sta=180.9,193.9
XS Rating Curve= 0 ,0
Exp/Cntr=0.3,0.1

Type RM Length L Ch R = 1 ,17665   ,178.9,174.1,168.6
XS GIS Cut Line= 3
     1858406.002      361734.025     1858369.534      361872.091
     1858504.998      362092.644
#Sta/Elev= 30
       0 1597.49     9.5 1594.59      19 1593.44    76.2 1590.16    85.7 1588.99
    95.2 1586.18   104.7  1581.6   114.2 1576.34   123.8 1571.31   133.3 1567.28
   142.8 1565.15     1661562.322   171.6 1561.77   179.5 1562.27   190.7 1563.16
   200.3 1563.08   209.9 1562.38   229.1 1561.96   248.2 1561.04   257.8 1561.13
   267.4 1561.51   286.6 1561.35   296.2 1562.35   315.4 1567.11   324.9 1568.47
   344.1 1570.48   353.7 1571.66   382.5 1575.91     392 1577.75   401.6 1581.42
#Mann= 3 , 0 , 0
       0     .08       0     166    .045       0   179.5     .08       0
#XS Ineff= 2 , 0
                          195.75          1567.7
Permanent Ineff=
       F       F
Bank Sta=166,179.5
XS Rating Curve= 0 ,0
Exp/Cntr=0.3,0.1

Type RM Length L Ch R = 1 ,17490.9 ,132.3,120.5,108.5
XS GIS Cut Line= 3
     1858126.403      361965.875     1858217.578      361971.083
     1858378.237      362135.789
#Sta/Elev= 29
       0 1577.67    27.4 1573.73    45.7 1571.24    54.8  1570.1    73.1 1568.02
    91.3 1565.82   100.9 1563.58   110.5 1559.92   120.1 1556.42   126.9 1554.92
   129.7  1554.3   139.3 1554.94   158.4 1557.66     168 1558.28   177.6 1558.42
   187.2 1558.24   196.8 1556.66   206.4 1553.25     216 1550.78   225.5  1550.4
   235.1 1550.75   244.7 1552.19   254.3 1555.29   263.9 1558.21   273.5 1560.52
   292.6 1565.47   302.2 1567.38   311.8 1568.56   321.4 1569.38
#Mann= 3 , 0 , 0
       0     .08       0   126.9    .045       0   139.3     .08       0
#XS Ineff= 2 , 0
                          178.26         1563.24
Permanent Ineff=
       F       F
Bank Sta=126.9,139.3
XS Rating Curve= 0 ,0
Exp/Cntr=0.3,0.1

Type RM Length L Ch R = 1 ,17370.3 ,43.4,62.2,84.8
XS GIS Cut Line= 3
      1858086.06      362068.526     1858163.295      362098.632
     1858369.138      362155.354
#Sta/Elev= 30
       0 1590.11     9.2 1582.76    18.4 1577.08    27.6  1573.6    36.8 1571.71
    64.5 1567.26    73.7 1565.11    82.9 1561.03    92.6 1555.74     101 1552.89
   102.3 1552.45     112 1552.43     116 1553.02   121.7 1553.85   131.4 1554.96
   141.1 1555.48   150.8 1555.75   170.2 1556.52     180 1556.34   189.6 1554.88
   199.4 1552.63   209.1 1553.12   218.8 1555.82   228.5 1556.81   238.2 1558.11
   247.9 1560.12   267.3 1565.39     277  1567.3   286.7 1568.46   296.4 1569.37
#Mann= 3 , 0 , 0
       0     .08       0     101    .045       0     116     .08       0
#XS Ineff= 2 , 0
                           167.4         1566.33
Permanent Ineff=
       F       F
Bank Sta=101,116
XS Rating Curve= 0 ,0
Exp/Cntr=0.3,0.1

Type RM Length L Ch R = 1 ,17308.1 ,77,80.1,190.8
XS GIS Cut Line= 6
     1858068.299       362083.28      1858128.35      362112.258
      1858192.75      362213.477     1858200.809      362239.403
     1858166.488      362342.345       1858283.8        362375.6
#Sta/Elev= 30
       0 1600.53      19 1584.34    28.6 1577.22    38.1 1572.81    47.6 1570.58
    75.9 1566.18    85.1 1564.03    94.4 1560.37   103.6  1555.8   112.8 1552.08
     122 1550.45     1441550.103   168.2 1551.26   186.6 1551.35   204.8 1550.24
   222.8 1547.67   249.8 1545.21   258.5 1545.12   275.8 1546.76   284.4 1547.19
   293.9 1547.08   322.5 1545.03   341.2 1545.18     360 1546.61   369.4 1547.76
   378.8 1549.39   388.1 1552.12   397.5 1556.01   416.3 1565.29   444.4 1581.25
#Mann= 3 , 0 , 0
       0     .08       0     122    .045       0     144     .08       0
#XS Ineff= 2 , 0
                          181.58         1564.91
Permanent Ineff=
       F       F
Bank Sta=122,144
XS Rating Curve= 0 ,0
Exp/Cntr=0.3,0.1

Type RM Length L Ch R = 1 ,17228   ,171.6,150.9,17.7
XS GIS Cut Line= 6
     1858023.928       362114.02     1858083.979      362142.998
     1858148.379      362244.217     1858156.438      362270.143
     1858124.374      362371.869     1858265.479      362400.955
#Sta/Elev= 30
       0 1625.06      19 1609.23    47.6  1582.4    57.2 1575.64    66.7 1570.96
    75.9 1568.29    85.1 1566.63   103.6 1564.68   131.3 1559.04   140.5  1557.9
   149.7 1556.05   168.2 1546.96   172.2 1545.95   177.4 1544.63   186.6 1544.73
   195.7 1545.69   213.8 1547.14   291.4 1542.08   310.8 1542.26   320.5 1541.88
   330.1 1542.67   358.9 1541.06   387.7 1540.69   397.3 1541.29   406.9 1543.33
   416.5 1546.64   426.1 1550.71   435.7 1555.39   445.3 1560.64   464.5  1572.5
#Mann= 3 , 0 , 0
       0     .08       0   172.2    .045       0   195.7     .08       0
#XS Ineff= 2 , 0
                          214.79         1557.73
Permanent Ineff=
       F       F
Bank Sta=172.2,195.7
XS Rating Curve= 0 ,0
Exp/Cntr=0.3,0.1

Type RM Length L Ch R = 1 ,17077.1 ,53.8,54.5,55.3
XS GIS Cut Line= 3
     1857991.783      362348.268     1858216.106      362418.545
     1858274.321      362446.767
#Sta/Elev= 30
       0 1578.05     9.8  1575.2    19.6  1574.1    29.4 1573.54    39.2  1572.1
      49 1568.96    68.6 1561.21    78.4 1557.07    88.2    1552      98 1546.24
   107.7 1540.97     1151539.428   117.5  1538.9     1221539.445   137.1 1541.56
   146.9 1541.56   156.7 1540.01   176.3 1535.69   186.1 1534.77   195.9 1534.39
   205.7 1534.63   215.5 1536.73   225.3 1540.56   235.1 1545.21   244.3 1550.51
   253.6  1557.1   262.8 1564.35   281.3 1580.62   290.5 1588.36   299.8 1595.37
#Mann= 3 , 0 , 0
       0      .1       0     115    .045       0     122     .08       0
Bank Sta=115,122
XS Rating Curve= 0 ,0
Exp/Cntr=0.3,0.1

Type RM Length L Ch R = 1 ,17022.6 ,84,86.7,89.3
XS GIS Cut Line= 2
      1857959.74      362390.377     1858244.649      362490.578
#Sta/Elev= 29
       0  1582.9     9.7    1580    19.5 1578.97    29.2 1578.52      39    1577
    48.7 1573.13    58.4  1567.9    68.2 1562.88    77.9 1558.46    87.7 1554.15
    97.4 1549.77   116.9 1541.53   126.6 1537.85     1301537.281   136.4  1536.2
     1441537.236   146.1 1537.52   155.9 1539.25   165.6 1539.06   175.4 1537.32
   185.1 1535.08   194.8  1533.9   204.6 1533.63   214.3 1534.26   224.1 1537.18
   233.8 1542.61     263 1562.31   272.8 1568.84     302 1588.65
#Mann= 3 , 0 , 0
       0      .1       0     130    .045       0     144      .1       0
Bank Sta=130,144
XS Rating Curve= 0 ,0
Exp/Cntr=0.3,0.1

Type RM Length L Ch R = 1 ,16935.9 ,186,184.9,183.6
XS GIS Cut Line= 3
     1857961.877      362470.549     1858148.254      362561.433
     1858228.559      362586.243
#Sta/Elev= 30
       0 1577.94     9.4 1571.53    28.3 1558.33    37.7 1552.07    47.1 1546.55
    56.6 1542.29      66 1539.01    84.8 1533.59    89.4 1532.86    94.2 1532.09
   103.7 1532.77   113.1  1534.5   122.5 1535.78     132 1536.06   141.4 1535.46
   150.8 1534.42   160.2 1533.75   169.6 1533.68   179.1 1534.32   188.5 1536.33
   197.9 1539.57   207.4 1543.38   216.7  1547.4     226 1551.63   235.4 1556.16
   244.7 1560.98     254 1566.06   263.4  1571.4   282.1 1582.97   291.4  1589.1
#Mann= 3 , 0 , 0
       0      .1       0    89.4    .045       0   103.7     .08       0
Bank Sta=89.4,103.7
XS Rating Curve= 0 ,0
Exp/Cntr=0.3,0.1

Type RM Length L Ch R = 1 ,16751   ,164.3,164.7,165
XS GIS Cut Line= 2
     1857870.255      362637.702      1858148.32       362755.57
#Sta/Elev= 27
       0 1573.19    19.5 1558.58    29.2 1551.45      39 1545.29    48.7 1540.83
    58.4 1537.72    87.7 1529.08    97.4 1526.64   107.2 1525.95   111.31526.578
   116.9 1527.44   126.6 1529.42   136.4 1530.82   146.1 1531.31   155.9 1531.08
   175.4 1529.59   185.1 1529.28   194.8 1530.13   204.6  1532.6   214.3 1536.48
   224.1 1541.21   253.3 1556.55     263 1561.75   272.8 1567.17   282.5 1572.87
   292.3 1578.78     302 1584.78
#Mann= 3 , 0 , 0
       0      .1       0    97.4    .045       0   111.3      .1       0
Bank Sta=97.4,111.3
XS Rating Curve= 0 ,0
Exp/Cntr=0.3,0.1

Type RM Length L Ch R = 1 ,16586.2 ,101.9,104.3,106.6
XS GIS Cut Line= 3
     1857823.243      362793.915     1857997.262      362871.231
     1858064.347      362909.054
#Sta/Elev= 22
       0 1547.04     9.5 1544.01      19 1541.11    38.1 1535.57    57.1 1530.24
    76.2 1525.06    85.7 1522.68    89.91522.093    95.2 1521.36   104.7 1521.94
   114.2 1523.23   123.8 1524.19   133.3 1524.54   142.8 1524.62   152.3 1525.31
   161.9 1527.83   171.4  1532.2     200 1547.24   209.7 1552.55   219.3 1558.11
   238.6 1569.54   267.4 1586.78
#Mann= 3 , 0 , 0
       0      .1       0    89.9    .045       0   104.7     .08       0
Bank Sta=89.9,104.7
XS Rating Curve= 0 ,0
Exp/Cntr=0.3,0.1

Type RM Length L Ch R = 1 ,16481.9 ,368.7,369.1,369.1
XS GIS Cut Line= 3
     1857778.618      362876.973     1857955.597      362978.673
      1858023.64       362994.71
#Sta/Elev= 22
       0 1552.82     9.7 1548.53    29.2 1539.74      68  1521.8    77.8 1518.34
    82.61517.655    87.5 1516.96    97.2 1517.36   116.6    1519   126.4 1519.61
   136.1 1519.98   145.8 1520.57   155.5 1521.89   165.2 1524.21     175 1527.44
   184.7 1532.78   194.4 1539.52   204.1 1545.53   212.9 1550.29   230.3 1559.18
   239.1 1563.96     274 1584.23
#Mann= 3 , 0 , 0
       0      .1       0    82.6    .045       0    97.2     .08       0
Bank Sta=82.6,97.2
XS Rating Curve= 0 ,0
Exp/Cntr=0.3,0.1

Type RM Length L Ch R = 1 ,16112.8 ,335.6,329.5,323.1
XS GIS Cut Line= 2
     1857535.834      363157.602     1857849.722      363341.993
#Sta/Elev= 30
       0 1596.52     9.8  1589.2    29.5 1575.04    39.4 1568.29    49.2 1561.92
      59 1556.16    78.7 1546.01    88.6 1541.32    98.4 1537.07   108.2 1533.19
   127.9 1526.01   147.6 1519.57   177.1  1510.3   184.3 1509.05   186.9  1508.6
   196.3 1508.87   206.6 1510.26   216.5 1511.34   226.3 1511.78   236.1 1512.72
     246 1513.94   255.8 1514.65   285.3 1514.42   295.2 1514.51     305 1515.69
   314.8 1517.93   334.5 1523.28   344.4 1526.37   354.2  1530.1     364 1534.96
#Mann= 3 , 0 , 0
       0      .1       0   184.3    .045       0   196.3     .08       0
Bank Sta=184.3,196.3
XS Rating Curve= 0 ,0
Exp/Cntr=0.3,0.1

Type RM Length L Ch R = 1 ,15783.3 ,225.1,223.5,221.6
XS GIS Cut Line= 2
     1857408.994      363510.384     1857761.337      363601.809
#Sta/Elev= 30
       0 1560.43     9.8 1555.58    19.7 1550.97    39.4 1542.34    49.2 1538.17
      59 1534.14    68.9  1529.9    78.7 1525.38   108.2 1511.27   127.9 1502.26
   137.7 1498.57   145.9 1497.22   147.6 1496.94   157.4 1496.92   160.9 1497.14
   177.1 1498.21   186.9 1498.63   196.8 1498.88   206.6 1499.26   216.4 1500.05
   226.3 1500.97   236.1 1501.58   265.6 1502.32   275.5 1503.42   285.3 1506.43
   295.1 1510.94   324.7 1525.53   334.5 1530.48   354.2 1540.66     364 1545.44
#Mann= 3 , 0 , 0
       0      .1       0   145.9    .045       0   160.9     .08       0
Bank Sta=145.9,160.9
XS Rating Curve= 0 ,0
Exp/Cntr=0.3,0.1

Type RM Length L Ch R = 1 ,15559.8 ,144,141.3,138.5
XS GIS Cut Line= 2
     1857371.612      363741.535     1857729.976      363805.341
#Sta/Elev= 30
       0 1575.88    19.7 1565.78    29.5 1560.39    39.4 1554.22    49.2 1547.11
    68.9 1531.81    88.5 1516.21    98.4 1508.71   108.2 1502.14     118 1497.26
   127.9 1493.39   137.7 1490.29   139.21490.141   147.6 1489.31   153.2 1489.73
   157.4 1490.04   167.2  1491.7   177.1 1492.95   206.6 1493.74   216.4 1493.49
   265.6 1490.57   275.5 1490.17   285.3 1489.91   295.1 1490.07     305 1491.69
   314.8 1495.52   324.6 1500.56   334.5 1505.88   354.2  1516.8     364 1522.36
#Mann= 3 , 0 , 0
       0      .1       0   139.2    .045       0   153.2      .1       0
#XS Ineff= 2 , 0
                          203.72          1503.6
Permanent Ineff=
       F       F
Bank Sta=139.2,153.2
XS Rating Curve= 0 ,0
Exp/Cntr=0.3,0.1

Type RM Length L Ch R = 1 ,15418.5 ,314.2,333.3,351.2
XS GIS Cut Line= 3
     1857414.446      363902.425     1857651.298      363915.463
     1857699.942       363958.91
#Sta/Elev= 25
       0 1525.41      38 1503.74    47.4 1498.18    56.9 1492.21    66.4 1487.08
    72.7 1485.46    75.9 1484.64    85.4 1484.81    87.7 1485.19    94.9 1486.38
   104.4 1488.24   113.9 1489.32   123.4 1489.86   142.3 1491.91   151.8 1492.01
   180.3 1490.27   199.3 1489.46   208.7 1488.95   218.2 1488.74   227.7 1489.37
   237.2 1491.36   246.5 1496.06   283.8 1517.99   293.1 1523.33   302.4 1528.81
#Mann= 3 , 0 , 0
       0      .1       0    72.7    .045       0    87.7     .08       0
#XS Ineff= 2 , 0
                          148.18          1496.9
Permanent Ineff=
       F       F
Bank Sta=72.7,87.7
XS Rating Curve= 0 ,0
Exp/Cntr=0.3,0.1

Type RM Length L Ch R = 1 ,15085.2 ,277.9,270.4,262.6
XS GIS Cut Line= 2
     1857345.892      364107.382      1857501.32      364290.333
#Sta/Elev= 29
       0 1492.12     9.6 1489.95    19.2 1489.07    28.8  1488.3    38.4 1487.47
      48 1486.62    57.6  1485.7    67.2 1484.73    76.8 1483.74    86.4 1482.69
      96 1481.22   105.6 1478.01   115.2  1474.5   119.7 1473.62   120.71473.426
   124.8 1472.63   134.4 1473.42   134.7 1473.51     144 1476.21   153.6 1479.65
   163.2 1481.99   172.8 1486.08   182.4 1493.06     192 1500.86   201.6 1508.76
   211.2 1516.46   220.9 1523.93   230.5 1530.89   240.1 1536.12
#Mann= 3 , 0 , 0
       0      .1       0   120.7    .045       0   134.4     .08       0
Bank Sta=120.7,134.4
XS Rating Curve= 0 ,0
Exp/Cntr=0.3,0.1

Type RM Length L Ch R = 1 ,14814.7 ,225.3,214.8,204.1
XS GIS Cut Line= 2
     1857121.019      364316.536     1857339.838      364444.354
#Sta/Elev= 30
       0 1516.68     9.8 1512.09    19.5 1507.33    29.2 1502.58      39 1497.62
    48.7 1492.42    58.5 1486.96    68.2 1481.77      78 1477.85    87.7 1474.28
    97.5 1470.45   107.2 1467.58   109.8 1467.39   110.81467.315     117 1466.85
   124.8 1467.19   126.7 1467.27   136.4 1468.29   146.2 1469.31     156  1470.1
   165.7 1470.85   175.4 1471.57   185.2 1472.28   194.9 1472.81   204.7 1473.29
   214.4 1475.14   224.2 1478.82   233.9 1482.94   243.7 1485.85   253.4 1486.79
#Mann= 3 , 0 , 0
       0      .1       0   110.8    .045       0   124.8      .1       0
Bank Sta=110.8,124.8
XS Rating Curve= 0 ,0
Exp/Cntr=0.3,0.1

Type RM Length L Ch R = 1 ,14600   ,60.1,70.4,80.2
XS GIS Cut Line= 3
     1857114.281      364570.433     1857167.046      364584.116
     1857359.684       364595.86
#Sta/Elev= 29
       0 1515.59     9.1 1509.63    18.2 1502.25    27.3 1493.98    36.3 1485.62
    45.4 1478.27    54.5 1472.25    64.2 1467.12    73.8 1463.83    76.5 1463.58
    83.5 1462.93    91.5 1463.46    93.1 1463.56   102.8 1464.64   112.4 1465.65
   122.1 1466.34   131.7 1466.61   141.4 1466.64     151 1466.58   160.7 1466.44
   170.3  1466.3     180 1466.16   189.6 1466.03   199.3 1465.97   208.9 1466.08
   218.6 1466.84   228.2 1468.79   237.9 1471.44   247.5 1473.82
#Mann= 3 , 0 , 0
       0      .1       0    73.8    .045       0    93.1      .1       0
#XS Ineff= 2 , 0
       0                     190       0    1470
Permanent Ineff=
       F       F
Bank Sta=73.8,93.1
XS Rating Curve= 0 ,0
Exp/Cntr=0.3,0.1

Type RM Length L Ch R = 1 ,14529.6 ,111.4,111.3,111.2
XS GIS Cut Line= 2
     1857081.364      364599.737      1857303.09      364722.444
#Sta/Elev= 29
       0 1526.93     9.8 1521.07    19.5 1514.98    29.2 1508.05      39 1499.93
    48.7 1491.11    58.5 1482.62    68.2 1476.65      78  1472.9    87.7 1467.95
    97.5 1463.01    99.5  1462.6   107.2 1461.01   114.5 1461.47     117 1461.63
   126.7 1462.91   136.4  1463.5   146.2  1463.5     156 1463.47   165.7 1463.57
   175.4 1463.76   185.2 1464.01   194.9 1464.29   204.7 1464.59   214.4 1464.92
   224.2 1465.31   233.9 1465.75   243.7  1466.2   253.4 1466.66
#Mann= 3 , 0 , 0
       0      .1       0    99.5    .045       0     117      .1       0
Bank Sta=99.5,117
XS Rating Curve= 0 ,0
Exp/Cntr=0.3,0.1

Type RM Length L Ch R = 1 ,14418.3 ,119.5,124.3,128.6
XS GIS Cut Line= 2
     1857026.894      364696.819     1857249.195       364818.48
#Sta/Elev= 29
       0 1518.48     9.8 1510.66    19.5 1502.21    29.2 1493.38      39 1485.23
    48.7 1479.78    58.5 1476.42    68.2 1472.46      78  1465.9    87.7  1458.9
      93 1457.23    97.5 1455.82   107.2 1456.81     108 1456.97     117 1458.78
   126.7 1460.36   136.4 1460.91   146.2 1460.73     156 1460.43   165.7 1460.24
   175.4 1460.21   185.2 1460.43   194.9 1460.84   204.7 1461.32   214.4 1461.75
   224.2 1462.02   233.9 1462.12   243.7 1462.17   253.4 1462.21
#Mann= 3 , 0 , 0
       0      .1       0      93    .045       0     108     .08       0
Bank Sta=93,108
XS Rating Curve= 0 ,0
Exp/Cntr=0.3,0.1

Type RM Length L Ch R = 1 ,14294   ,383.5,385.3,385.9
XS GIS Cut Line= 2
     1856927.325      364744.794     1857206.056      364980.953
#Sta/Elev= 29
       0 1551.87    19.2 1537.68    38.5 1523.17    48.1 1515.74    57.7 1508.16
    76.9 1492.71    86.5 1485.84    96.1 1481.82   105.8 1479.66   115.4 1477.37
     125 1473.28   134.6 1467.89   153.8 1455.49   161.7 1452.18   163.4 1451.47
     173 1451.25     1771452.029   182.7 1453.15   192.3 1455.56   201.9 1456.47
   211.5 1456.56   269.2 1456.34   278.8 1456.69     298 1457.98   307.6  1458.4
   336.5  1458.6   346.1 1458.85   355.7 1460.64   365.3 1464.51
#Mann= 3 , 0 , 0
       0      .1       0   161.7    .045       0     177      .1       0
Bank Sta=161.7,177
XS Rating Curve= 0 ,0
Exp/Cntr=0.3,0.1

Type RM Length L Ch R = 1 ,13908.7 ,428.7,416,402.2
XS GIS Cut Line= 2
      1856712.91      365034.627     1856980.107       365282.22
#Sta/Elev= 30
       0 1542.14    38.3 1508.98    47.9  1500.9    57.5  1493.9    67.1 1489.21
    76.7 1487.23    86.3 1485.99    95.9 1483.72   105.4 1479.96     115 1475.32
   134.2 1465.56   143.8 1460.57   153.4 1455.39     163 1449.23   172.6 1442.66
     181 1438.52   182.1 1437.98   191.7 1437.68     196 1438.42   201.3 1439.34
   220.5 1444.23   230.1 1446.12   239.7 1447.58   249.2 1448.86   258.8 1449.86
     278 1451.19   287.6 1453.14   297.2 1456.03   316.3 1462.72   364.3 1479.15
#Mann= 3 , 0 , 0
       0      .1       0     181    .045       0     196      .1       0
Bank Sta=181,196
XS Rating Curve= 0 ,0
Exp/Cntr=0.3,0.1

Type RM Length L Ch R = 1 ,13492.7 ,395.5,391.5,386.7
XS GIS Cut Line= 2
     1856452.149      365478.509     1856811.476      365536.939
#Sta/Elev= 30
       0 1504.68     9.8  1499.6    19.7 1496.83    49.2 1493.43    68.9 1491.47
    78.7 1489.77    88.6 1485.79    98.4 1479.94   137.8 1455.02   147.6 1447.74
   157.4 1438.86   167.3 1431.59   174.4 1429.57   177.1  1428.8   186.9 1428.67
     1931429.206   206.6 1430.96   216.5 1432.81   226.3 1435.77     246  1443.8
   255.8 1447.02   265.7 1449.41   275.5 1451.07   295.2 1453.48     305  1454.3
   324.7 1455.32   334.5 1456.36   344.4 1457.78   354.2  1459.6     364  1463.1
#Mann= 3 , 0 , 0
       0      .1       0   174.4    .045       0     193      .1       0
Bank Sta=174.4,193
XS Rating Curve= 0 ,0
Exp/Cntr=0.3,0.1

Type RM Length L Ch R = 1 ,13101.2 ,224.6,238.9,252.2
XS GIS Cut Line= 3
     1856463.923      365848.974     1856513.339       365880.36
     1856807.195      365865.735
#Sta/Elev= 30
       0 1485.23     9.8 1481.39    19.5 1475.28    29.3 1468.23      39 1461.07
    48.8 1454.32    58.5 1448.38    68.4  1443.1      88 1433.06    97.8 1428.31
   107.6 1424.97   117.4 1423.72   127.2 1423.52     137 1423.05   146.8 1421.85
   166.4 1417.18     1681417.056   176.2 1416.43     182  1417.3   185.8 1417.87
   195.8 1421.18   205.6 1424.59   215.5 1426.84   225.3 1428.23   274.3 1433.28
   284.1 1434.19   303.7 1435.46   313.5 1437.32   323.3 1440.35   352.8 1450.62
#Mann= 3 , 0 , 0
       0      .1       0     168    .045       0     182      .1       0
Bank Sta=168,182
XS Rating Curve= 0 ,0
Exp/Cntr=0.3,0.1

Type RM Length L Ch R = 1 ,12862.3 ,133.1,154.1,174.4
XS GIS Cut Line= 2
     1856420.378      366011.868     1856739.117      366212.395
#Sta/Elev= 30
       0 1455.52    19.3 1445.78      29 1441.04    38.6 1436.78    48.3  1432.9
    67.6  1424.9    77.2 1421.07    86.9 1418.25    96.6 1416.89   106.2 1416.31
   115.9 1415.54   125.5 1414.47   135.2 1413.22   144.8 1411.72   154.1 1410.44
   164.2 1410.19   169.1 1410.56   173.8 1410.91   193.1  1413.4   212.4 1415.56
   222.1 1416.54   231.7 1417.33   241.4 1417.98     251 1419.63   260.7  1423.3
   270.4 1428.91   318.6 1457.88     338 1469.67   357.3 1481.77   376.6 1494.58
#Mann= 3 , 0 , 0
       0      .1       0   154.1    .045       0   169.1      .1       0
Bank Sta=154.1,169.1
XS Rating Curve= 0 ,0
Exp/Cntr=0.3,0.1

Type RM Length L Ch R = 1 ,12708.2 ,332.1,322.2,311
XS GIS Cut Line= 4
     1856385.777      366043.481     1856446.056      366136.446
     1856460.462      366268.471     1856516.032      366363.892
#Sta/Elev= 30
       0 1458.24    18.5 1448.87    27.7  1444.1    36.9 1439.54    46.2  1435.6
    73.9 1425.45    83.1 1421.99    92.3 1418.66   101.6 1416.35   110.8 1415.24
   120.3 1414.54   139.3 1413.36   148.7 1412.36   158.2 1410.65   167.7 1408.39
   177.2 1406.53   186.7 1406.25     1891406.541   196.2 1407.46   205.7 1409.56
   215.2 1411.51   224.6  1412.6   234.1 1413.29   243.6 1415.36   252.8 1420.57
     262 1427.25   317.2 1469.25   326.4 1476.07   335.6 1482.33     354 1493.92
#Mann= 3 , 0 , 0
       0      .1       0   177.2    .045       0     189     .08       0
Bank Sta=177.2,189
XS Rating Curve= 0 ,0
Exp/Cntr=0.3,0.1

Type RM Length L Ch R = 1 ,12386.1 ,265.4,256.9,247.9
XS GIS Cut Line= 2
     1856068.433      366098.332     1856264.683      366414.892
#Sta/Elev= 30
       0  1496.9     9.8  1488.7    19.6  1479.5    39.2  1459.9      49 1450.68
    58.8 1442.46    68.6 1435.52    78.4 1429.24    88.2 1423.56      98 1418.43
   117.6 1410.01   137.2 1401.06     147 1397.39   149.5 1396.97   156.8 1395.74
   166.6 1396.24   186.2 1399.43     196 1400.88   225.4 1404.73     245 1406.99
   254.8 1406.97   274.4    1405   284.2  1404.7     294 1405.04   303.8 1405.55
   323.4 1406.61   333.2 1407.37     343 1408.44   352.8 1409.89   372.5 1413.85
#Mann= 3 , 0 , 0
       0      .1       0   149.5    .045       0   166.6      .1       0
Bank Sta=149.5,166.6
XS Rating Curve= 0 ,0
Exp/Cntr=0.3,0.1

Type RM Length L Ch R = 1 ,12129.1 ,379.1,379.2,379.1
XS GIS Cut Line= 3
     1855856.277       366328.03     1856003.469      366435.075
     1856150.661      366542.119
#Sta/Elev= 25
       0 1495.92    19.2 1483.07    28.7 1476.59    57.5 1457.16   105.4 1423.86
     115 1417.28   124.5 1411.25   134.1 1406.75   143.7 1404.58   162.8 1401.96
   172.4 1400.02   190.51394.336   191.6 1393.99   201.2 1393.48   204.51394.453
   210.7 1396.29   220.3 1400.07   229.9  1402.4   239.5 1402.94   277.8  1403.6
   325.7 1404.29   335.3 1404.88   344.8 1407.36   354.4 1410.85     364  1413.9
#Mann= 3 , 0 , 0
       0      .1       0   190.5    .045       0   204.5     .08       0
Bank Sta=190.5,204.5
XS Rating Curve= 0 ,0
Exp/Cntr=0.3,0.1

Type RM Length L Ch R = 1 ,11749.9 ,266,262.1,257.8
XS GIS Cut Line= 3
     1855668.723      366659.735     1855815.915       366766.78
     1855963.107      366873.824
#Sta/Elev= 30
       0 1470.16    38.3 1445.16    57.5 1432.41    86.2 1412.45    95.8 1405.89
   105.4 1399.81     115 1394.98   124.5 1390.67   134.1 1387.02   137.21386.382
   143.7 1385.04   153.3 1385.52   156.21386.348   172.4 1391.05     182 1392.17
   191.6 1392.09   239.5 1389.82     249 1389.49   258.6 1389.32   268.2 1389.42
   277.8 1389.76   287.4 1390.29     297 1391.26   306.5 1393.15   316.1 1395.61
   325.7 1397.46   335.3 1398.46   344.8 1401.05   354.4 1405.26     364 1410.19
#Mann= 3 , 0 , 0
       0      .1       0   137.2    .045       0   156.2     .08       0
#XS Ineff= 2 , 0
                           193.8         1400.66
Permanent Ineff=
       F       F
Bank Sta=137.2,156.2
XS Rating Curve= 0 ,0
Exp/Cntr=0.3,0.1

Type RM Length L Ch R = 1 ,11487.8 ,210.1,199.5,188.2
XS GIS Cut Line= 2
     1855504.425      366896.279     1855832.608      367054.184
#Sta/Elev= 23
       0 1469.93    19.2 1457.34    38.3 1444.93    57.5  1432.8    76.7  1421.2
    95.8 1409.97   105.4 1404.08     115  1397.4   124.6 1389.47   134.2 1382.13
   140.8 1379.72   143.8 1378.63   153.4 1378.66   159.81379.542   172.5 1381.47
   182.1 1382.45   191.7 1382.92   210.8 1383.62   287.5 1386.18   325.9 1387.56
     345 1388.03   354.6  1388.4   364.2 1389.74
#Mann= 3 , 0 , 0
       0      .1       0   140.8    .045       0   159.8     .08       0
Bank Sta=140.8,159.8
XS Rating Curve= 0 ,0
Exp/Cntr=0.3,0.1

Type RM Length L Ch R = 1 ,11288.3 ,212.2,224.7,237.4
XS GIS Cut Line= 3
     1855507.044      367077.677     1855538.266       367152.98
     1855787.117      367144.255
#Sta/Elev= 23
       0 1417.06    18.1 1409.75    36.2 1402.63    45.3 1399.53    54.4 1397.16
    81.5 1390.85    91.1 1390.69   100.7 1390.08   110.2 1388.47   119.8  1385.6
   129.4 1381.82     139 1377.48   148.6    1374   158.1 1372.79   167.7 1374.22
   177.3  1377.4   186.9 1379.75   196.4 1380.56   282.6 1383.32   301.8 1383.81
   311.4 1384.19     321 1385.39   330.5 1388.01
#Mann= 3 , 0 , 0
       0      .1       0   148.6    .045       0   167.7     .08       0
Bank Sta=148.6,167.7
XS Rating Curve= 0 ,0
Exp/Cntr=0.3,0.1

Type RM Length L Ch R = 1 ,11063.6 ,135.5,143.7,151.8
XS GIS Cut Line= 2
     1855384.879      367269.598     1855700.124      367451.579
#Sta/Elev= 27
       0 1459.66     9.8 1454.99    19.7 1450.38    29.5 1445.84    39.4 1441.36
      59  1432.6    88.5 1420.14    98.4 1415.46   108.2 1409.68   127.9 1396.53
   137.7 1389.68   147.6 1382.11   157.4 1374.21   163.4 1370.84   167.2  1368.7
   177.1 1368.11     1801368.959   186.9 1370.98   196.8 1373.38   206.6 1374.08
   275.5 1374.29   314.8 1374.98   324.6 1375.39   334.5 1377.74   344.3 1382.53
   354.2 1388.33     364  1394.3
#Mann= 3 , 0 , 0
       0      .1       0   163.4    .045       0     180     .08       0
Bank Sta=163.4,180
XS Rating Curve= 0 ,0
Exp/Cntr=0.3,0.1

Type RM Length L Ch R = 1 ,10920   ,576.8,555.4,533.8
XS GIS Cut Line= 2
     1855364.448      367372.352     1855595.001      367654.078
#Sta/Elev= 21
       0 1440.47    29.5 1423.43    39.4  1417.8    49.2 1412.06      59 1405.57
    68.9 1398.39    78.7  1390.9    88.6 1383.02    98.4 1373.98   108.2 1367.02
   108.5 1366.95   118.1 1364.55   127.9 1366.65   137.7 1369.63   147.6 1370.81
   157.4 1370.98   196.8 1371.05     305  1371.5   344.4 1371.59   354.2 1372.34
     364  1376.1
#Mann= 3 , 0 , 0
       0      .1       0   108.5    .045       0   127.9     .08       0
Bank Sta=108.5,127.9
XS Rating Curve= 0 ,0
Exp/Cntr=0.3,0.1

Type RM Length L Ch R = 1 ,10364.6 ,126.9,137,146.6
XS GIS Cut Line= 2
     1855035.811      367939.125     1855399.059      367915.415
#Sta/Elev= 24
       0 1430.92     9.8 1424.49    19.7 1418.32    29.5 1412.35      59  1394.7
    98.4 1370.66   108.2 1364.34   118.1 1357.54   127.9 1352.33   137.7 1350.67
   147.6 1352.12   157.4 1355.36   167.2  1357.9   177.1 1358.59   226.3 1358.82
   275.5 1358.46   285.3 1358.27   295.2 1357.87     305  1357.2   314.8 1356.88
   324.7  1357.5   334.5 1359.56   344.3 1363.63     364 1374.07
#Mann= 3 , 0 , 0
       0      .1       0   127.9    .045       0   147.6     .08       0
Bank Sta=127.9,147.6
XS Rating Curve= 0 ,0
Exp/Cntr=0.3,0.1

Type RM Length L Ch R = 1 ,10227.6 ,118.6,122.1,125.4
XS GIS Cut Line= 3
     1855013.082      368013.229     1855373.794      368153.003
     1855417.765      368152.077
#Sta/Elev= 30
       0 1438.04     9.7 1432.09    19.3 1425.97      29 1419.65    48.4 1406.83
    77.4 1387.38   106.4 1367.58     116 1360.19   125.7 1352.98   135.3 1348.47
   145.1 1347.63   150.3 1348.42   164.4 1350.55   174.1 1350.98   212.8 1351.43
   232.1 1351.44   241.8 1351.34   251.4 1351.06   261.1 1350.53   280.5 1348.74
   290.1 1348.16   309.5 1347.82   338.5 1347.03   348.2 1347.16   357.8 1347.85
   377.2 1349.63   386.8 1351.16   395.6 1353.95   404.4 1358.32   430.8 1373.69
#Mann= 3 , 0 , 0
       0      .1       0   135.3    .045       0   150.3     .08       0
#XS Ineff= 2 , 0
                          218.78         1359.64
Permanent Ineff=
       F       F
Bank Sta=135.3,150.3
XS Rating Curve= 0 ,0
Exp/Cntr=0.3,0.1

Type RM Length L Ch R = 1 ,10105.5 ,256.3,260.3,264.6
XS GIS Cut Line= 2
     1854984.563      368112.529     1855331.803      368310.983
#Sta/Elev= 30
       0 1430.44     9.8 1424.57    19.5 1417.77    29.3 1410.02    48.8 1393.41
    68.3 1376.28      78 1367.39    87.8 1357.61    97.6 1348.84   107.3 1344.41
   107.5  1344.4   117.1 1344.08   122.5 1344.66   126.8 1345.12   136.6 1345.77
   214.6  1347.1   224.4 1347.22   234.1 1347.08   243.9 1346.36   263.4 1344.01
   273.1 1343.19   292.6 1342.66   312.2  1341.6   321.9 1341.38   331.7 1342.07
   351.2 1345.81   360.9 1348.12   370.7 1351.08   380.4 1354.77     400 1362.76
#Mann= 3 , 0 , 0
       0      .1       0   107.5    .045       0   122.5     .06       0
#XS Ineff= 2 , 0
       0                   224.4       0 1359.77
Permanent Ineff=
       F       F
Bank Sta=107.5,122.5
XS Rating Curve= 0 ,0
Exp/Cntr=0.3,0.1

Type RM Length L Ch R = 1 ,9845.2  ,214,207.7,201
XS GIS Cut Line= 4
     1854815.691      368257.529     1854916.766      368364.679
     1855010.472      368443.987     1855119.612      368569.254
#Sta/Elev= 30
       0 1429.71    29.5 1413.09    49.1 1401.79    78.6 1384.35     108 1366.53
   117.8 1360.86   127.7 1355.56   137.5 1350.87   147.3 1346.98   156.7 1343.62
   166.2 1340.36   175.6 1337.64   179.4 1337.17   185.1 1336.47   194.4 1336.85
   213.4 1339.51   260.6 1341.84   270.1 1342.25   279.8 1342.44   289.6  1341.8
   299.4 1340.23   318.9 1335.99   328.7 1334.41   338.5 1333.35   348.2 1334.06
     358 1338.46   377.6 1352.08   397.1 1365.09   416.7 1378.36   436.2 1391.97
#Mann= 3 , 0 , 0
       0      .1       0   179.4    .045       0   194.4      .1       0
#XS Ineff= 2 , 0
                          272.81         1351.22
Permanent Ineff=
       F       F
Bank Sta=179.4,194.4
XS Rating Curve= 0 ,0
Exp/Cntr=0.3,0.1

Type RM Length L Ch R = 1 ,9637.5  ,116.2,122.3,128.4
XS GIS Cut Line= 2
     1854776.779       368540.08     1855047.101      368659.089
#Sta/Elev= 30
       0  1365.5    19.1 1353.14    28.6 1347.14    38.1  1341.4    47.6 1336.03
    57.2 1331.89    59.7  1331.6    66.7 1330.79    74.7 1331.58    76.2 1331.73
    85.8 1333.21    95.3 1333.99   104.8 1334.19   123.9  1334.2   133.4 1334.09
   142.9 1333.85   152.4 1333.46     162 1332.92   171.5 1332.22     181 1331.27
   190.6 1330.47   200.1  1330.8   209.6 1332.83   219.1 1335.88   228.7 1340.25
   238.2 1345.89   266.8 1364.06   276.3 1370.41   285.8 1377.05   295.4 1383.92
#Mann= 3 , 0 , 0
       0      .1       0    59.7    .045       0    74.7     .08       0
#XS Ineff= 2 , 0
                          117.45         1339.95
Permanent Ineff=
       F       F
Bank Sta=59.7,74.7
XS Rating Curve= 0 ,0
Exp/Cntr=0.3,0.1

Type RM Length L Ch R = 1 ,9515.2  ,595.4,595.1,594.9
XS GIS Cut Line= 2
     1854677.361      368593.389      1854959.64      368823.203
#Sta/Elev= 30
       0 1387.13     9.8 1384.58    19.7 1382.14    29.5 1379.47    39.4 1374.63
    49.2 1368.23    68.9 1353.94    88.5 1339.23    98.4 1332.27   108.2 1327.26
   108.6 1327.22     118 1326.34   123.6 1327.03   127.9 1327.56   137.7  1329.1
   147.6 1329.76   177.1 1329.76   206.6 1329.53   216.4 1329.01   236.1 1326.51
     246 1326.54   255.8 1328.06   265.6 1330.09   275.5 1332.32   285.3 1335.08
   295.1 1338.74     305 1343.17   314.8 1348.38   324.6 1353.99     364  1378.8
#Mann= 3 , 0 , 0
       0      .1       0   108.6    .045       0   123.6     .08       0
Bank Sta=108.6,123.6
XS Rating Curve= 0 ,0
Exp/Cntr=0.3,0.1

Type RM Length L Ch R = 1 ,8920.1  ,159.8,161.5,163.1
XS GIS Cut Line= 3
     1854296.621      369052.374     1854534.213      369241.773
     1854587.085       369269.79
#Sta/Elev= 25
       0 1382.46      49 1351.63    88.2 1327.15      98 1320.97   107.8 1314.59
   117.6 1309.74   118.5 1309.62   127.4 1308.39   133.5 1309.43   137.2 1310.06
     147 1311.95   156.8 1312.76   166.6 1313.07   176.4 1313.26   186.2 1313.19
   205.8 1312.33   215.6 1312.25   284.2  1313.9     294 1314.61   303.8 1316.55
   312.4 1320.33   320.9 1324.78   329.5 1329.43   355.1  1343.5   363.7 1348.11
#Mann= 3 , 0 , 0
       0      .1       0   118.5    .045       0   133.5     .08       0
Bank Sta=118.5,133.5
XS Rating Curve= 0 ,0
Exp/Cntr=0.3,0.1

Type RM Length L Ch R = 1 ,8758.6  ,68.7,68.6,68.7
XS GIS Cut Line= 3
     1854232.805      369200.763     1854449.986      369401.215
      1854567.55      369416.972
#Sta/Elev= 30
       0 1347.43    28.6 1330.05    38.1 1323.77    47.7 1316.04    57.2 1308.56
    66.7 1305.13    76.3 1304.68    81.11305.393    95.3 1307.51   104.9 1308.59
   133.5 1309.21   152.5 1309.13   162.1 1309.35   181.1 1310.26   247.9 1313.09
   276.5 1314.46     286 1315.18   295.6 1316.08   304.7 1318.03   313.8 1321.52
   322.9 1326.04     332 1330.15   341.2 1333.33   350.3 1336.33   359.4 1339.16
   368.5 1341.32   377.7 1342.95   386.8 1344.13   395.9 1345.02   414.2 1346.37
#Mann= 3 , 0 , 0
       0      .1       0    66.7    .045       0    81.1     .08       0
Bank Sta=66.7,81.1
XS Rating Curve= 0 ,0
Exp/Cntr=0.3,0.1

Type RM Length L Ch R = 1 ,8690    ,281.2,277.3,272.9
XS GIS Cut Line= 3
     1854183.311      369247.654     1854417.764      369461.259
     1854447.723      369600.625
#Sta/Elev= 30
       0    1344    38.4 1321.07    48.1 1315.55    57.7 1311.41    67.3    1308
    76.9 1305.33    79.3 1305.05    86.5  1304.2    96.1 1304.91   115.3 1308.17
   124.9 1308.28   153.8 1307.87   163.4  1308.1   192.2 1309.51   259.5 1313.46
   288.3 1314.56     298 1315.42   307.6 1317.01   317.2 1318.86   326.7  1321.6
   336.2 1325.11   345.7 1329.06   355.2 1333.49   364.7 1338.25   374.2 1343.54
   383.7  1349.2   421.7 1373.31   440.7 1384.92   450.2 1390.36   459.7 1394.76
#Mann= 3 , 0 , 0
       0      .1       0    79.3    .045       0    96.1     .08       0
Bank Sta=79.3,96.1
XS Rating Curve= 0 ,0
Exp/Cntr=0.3,0.1

Type RM Length L Ch R = 1 ,8412.7  ,372,372.1,371.3
XS GIS Cut Line= 2
     1853931.833      369428.507     1854239.401      369623.593
#Sta/Elev= 23
       0 1394.51    28.8 1376.32    38.3 1370.25    67.1  1352.2    95.8 1334.32
   124.6 1316.69   134.2 1311.26   143.8 1306.66   153.4 1302.81   162.9 1300.13
   172.5 1299.55   177.3 1300.04   182.1 1300.52   191.7 1301.75   201.3 1302.38
   239.6 1302.47   249.2 1302.68   258.8 1303.11     278 1304.34   335.5 1308.23
     345 1309.37   354.6 1311.89   364.2 1316.22
#Mann= 3 , 0 , 0
       0      .1       0   162.9    .045       0   177.3     .08       0
Bank Sta=162.9,177.3
XS Rating Curve= 0 ,0
Exp/Cntr=0.3,0.1

Type RM Length L Ch R = 1 ,8040.7  ,122.4,93.1,5.7
XS GIS Cut Line= 3
     1853761.576       369676.79     1853864.388      369801.133
     1854070.705      369928.253
#Sta/Elev= 30
       0 1342.42      19  1333.3    28.5 1328.95    47.4 1320.56    56.9 1316.53
    66.4  1312.7    75.9 1309.68    85.4 1308.17    94.9 1307.84   123.4 1307.49
   132.9 1307.09   142.4 1305.71   151.8 1302.96     171 1295.22   180.7  1292.6
   190.4 1291.52   216.91290.036   219.5 1289.92   229.2 1290.02   238.9 1290.91
   248.6 1292.34   258.3 1293.45     268 1293.83   277.7 1293.96   316.4 1295.06
   326.1 1295.98   335.8 1298.86   345.5 1305.29   355.2 1313.02   403.7 1353.25
#Mann= 3 , 0 , 0
       0      .1       0   216.9    .045       0   229.2     .08       0
#XS Ineff= 2 , 0
       0                     250       0    1300
Permanent Ineff=
       F       F
Bank Sta=216.9,229.2
XS Rating Curve= 0 ,0
Exp/Cntr=0.3,0.1

Type RM Length L Ch R = 1 ,7947.5  ,98.2,79.2,132.7
XS GIS Cut Line= 6
     1853585.829      369849.764      1853735.96      369999.785
     1853813.067      369946.643     1853888.089      369891.937
     1853932.374      369849.214     1854079.042      369976.185
#Sta/Elev= 30
       0 1324.36    19.3  1316.5    28.9  1312.8    38.6 1310.06    57.9 1305.42
    96.5  1294.6   106.1 1292.35   115.8 1291.01   154.4 1289.98   212.2 1288.97
   249.7 1289.23   324.5 1290.75   333.7 1290.69   352.3 1289.14   361.2 1288.76
   370.9 1288.66   380.2 1288.74   416.3 1290.27   460.3 1291.74     470 1292.98
   479.7 1293.57   499.1 1293.94   537.9 1295.33   547.6 1296.92   557.3 1301.16
     567 1308.31   586.4 1324.73   634.9  1366.7   644.6 1374.55   654.3 1381.15
#Mann= 3 , 0 , 0
       0     .08       0   361.2    .045       0   380.2     .08       0
Bank Sta=361.2,380.2
XS Rating Curve= 0 ,0
Exp/Cntr=0.3,0.1

Type RM Length L Ch R = 1 ,7868.4  ,82.7,118.8,140.6
XS GIS Cut Line= 6
     1853580.272      369869.214     1853759.406      370056.921
     1853836.513      370003.778     1853911.535      369949.072
     1853955.819       369906.35     1854058.897      369999.803
#Sta/Elev= 30
       0 1321.12    28.8 1309.81    38.4 1306.82    67.3 1300.17    86.5 1294.81
    96.1 1292.44   105.7 1291.15   134.5 1289.98   201.8 1288.39     221 1288.41
   259.5 1289.02   287.6 1288.44   334.4 1288.86   343.8 1288.71   362.4 1287.12
   371.7 1286.77   384.51287.039   390.2 1287.37   418.1 1290.55   427.4 1291.25
     446 1292.03     526 1294.43   535.3 1294.92   544.6 1296.19   553.9 1300.82
   563.2 1307.84     591 1332.26   628.1 1365.69   637.4 1373.42   646.6 1380.01
#Mann= 3 , 0 , 0
       0     .08       0   362.4    .045       0   384.5     .08       0
Bank Sta=362.4,384.5
XS Rating Curve= 0 ,0
Exp/Cntr=0.3,0.1

Type RM Length L Ch R = 1 ,7749.6  ,51.7,72.4,92.2
XS GIS Cut Line= 4
     1853576.104      369878.245     1853765.751      370086.641
       1853850.5      370089.418      1853935.25      370166.525
#Sta/Elev= 30
       0 1320.13    29.2 1308.78    38.9 1305.61    48.6 1302.92      68 1298.88
    87.4 1293.72    97.2 1291.72   106.9 1290.77   126.3 1289.98   184.6 1288.29
     204 1287.97   233.2 1288.61   262.3 1290.07   281.8 1291.29   291.2 1290.59
   307.8 1286.64     310 1286.12   319.5 1285.56   324.81286.408   328.9 1287.06
   338.3 1290.04   347.7  1292.7   357.1  1294.1   366.6 1294.87   376.1 1296.91
   385.7 1301.59   414.3 1321.27   452.5 1346.72   471.6 1360.09   481.1 1366.42
#Mann= 3 , 0 , 0
       0     .08       0   307.8    .045       0   324.8      .1       0
Bank Sta=307.8,324.8
XS Rating Curve= 0 ,0
Exp/Cntr=0.3,0.1

Type RM Length L Ch R = 1 ,7677.3  ,160.3,166.8,173.3
XS GIS Cut Line= 3
     1853552.916      369958.826     1853744.385      370119.029
     1853839.469      370245.369
#Sta/Elev= 30
       0 1304.68     9.6 1301.61    28.8 1297.12    38.4 1295.08      48 1293.34
    67.2 1290.69    76.8 1289.57    86.4 1288.91   153.6  1287.1   172.8 1287.22
     192 1287.96   220.8  1289.7   249.6 1291.72     259 1291.93   268.2 1290.49
   277.6 1287.34   283.3 1285.71   286.9 1284.68   296.2  1284.8   298.3 1285.71
   305.5 1288.81   314.8 1295.89   324.1  1303.6   333.4 1310.96   342.7 1318.73
     352 1326.94   370.6  1344.7   379.9 1352.55   389.2    1359   407.8 1369.77
#Mann= 3 , 0 , 0
       0     .08       0   283.3    .045       0   298.3      .1       0
Bank Sta=283.3,298.3
XS Rating Curve= 0 ,0
Exp/Cntr=0.3,0.1

Type RM Length L Ch R = 1 ,7510.4  ,218.8,207.4,195.8
XS GIS Cut Line= 3
     1853472.162      370014.834     1853612.835      370201.088
     1853674.054      370365.202
#Sta/Elev= 29
       0 1316.29    19.4 1305.84    29.2 1300.68    38.9 1296.48    48.6 1293.91
    58.4 1292.73     107 1287.81   126.4 1285.94   136.2 1285.34   145.9 1285.14
   155.6 1285.31   194.5 1286.82   233.4 1288.59   243.1 1288.25   252.9  1285.8
   260.9 1282.81   262.6 1282.17   272.3 1281.21   275.9 1282.52   282.1 1284.78
   291.8 1294.03   301.5 1303.84     321 1320.55   330.7 1328.71   340.4 1336.66
   350.2 1344.14   359.9 1350.46   369.6 1355.48   408.6 1373.93
#Mann= 3 , 0 , 0
       0     .08       0   260.9    .045       0   275.9      .1       0
Bank Sta=260.9,275.9
XS Rating Curve= 0 ,0
Exp/Cntr=0.3,0.1

Type RM Length L Ch R = 1 ,7303    ,187.3,188.6,189.5
XS GIS Cut Line= 2
     1853302.129      370222.214     1853579.296      370458.168
#Sta/Elev= 26
       0 1293.67     9.8 1288.48    19.7 1284.45    29.5 1282.69    39.4 1282.06
      59    1281    68.9 1280.59    78.7 1280.52    98.4 1280.76   177.1 1282.08
   186.9 1282.13   196.8 1281.26   206.6 1278.34   211.4 1277.15   216.4 1275.91
   226.3 1276.89   236.1 1281.88     246 1290.11   255.8 1297.67   265.6 1304.53
     305 1330.77   314.8  1337.4   324.6 1343.78   334.5  1349.3   344.3 1354.48
     364 1364.73
#Mann= 3 , 0 , 0
       0     .08       0   211.4    .045       0   226.3      .1       0
Bank Sta=211.4,226.3
XS Rating Curve= 0 ,0
Exp/Cntr=0.3,0.1

Type RM Length L Ch R = 1 ,7114.4  ,205.2,217.9,230.2
XS GIS Cut Line= 2
      1853185.84      370352.122     1853450.722      370601.788
#Sta/Elev= 28
       0 1280.04     9.8 1278.67    29.5 1277.76    39.4 1277.47      59 1277.18
    78.7 1276.67    98.4 1276.59   127.9 1276.32   147.6 1276.35   177.1 1276.74
   186.9  1277.1   206.6 1278.66   216.4 1279.03   226.3 1276.86   236.1 1273.52
   238.6 1272.99     246 1271.44   252.6  1272.9   255.8 1273.61   265.6 1280.55
   275.5 1288.94   285.3 1296.62   295.1 1303.81   324.6 1325.14   334.5 1331.89
   344.3 1337.59   354.2 1342.34     364  1346.8
#Mann= 3 , 0 , 0
       0     .08       0   238.6    .045       0   252.6      .1       0
#XS Ineff= 2 , 0
          214.35 1287.93
Permanent Ineff=
       F       F
Bank Sta=238.6,252.6
XS Rating Curve= 0 ,0
Exp/Cntr=0.3,0.1

Type RM Length L Ch R = 1 ,6896.5  ,145.8,140.6,135.3
XS GIS Cut Line= 2
     1853140.622      370445.818     1853235.445       370797.25
#Sta/Elev= 28
       0 1275.31    19.7 1274.85    29.5 1274.79      59 1274.88   127.9 1274.92
   147.6  1274.7   157.4  1274.4   167.2 1273.95   177.1 1273.36   186.9 1272.31
   196.8 1269.73   206.6 1266.11   213.3 1264.84   216.4 1264.25   226.3 1264.21
   228.3 1264.66   236.1 1266.41     246 1272.94   255.8 1281.65   265.6 1289.22
   275.5 1296.12   285.3 1302.17   295.1 1306.49     305 1309.28   314.8 1310.63
   324.6 1311.27   354.2 1312.12     364  1313.1
#Mann= 3 , 0 , 0
       0     .08       0   213.3    .045       0   228.3     .08       0
Bank Sta=213.3,228.3
XS Rating Curve= 0 ,0
Exp/Cntr=0.3,0.1

Type RM Length L Ch R = 1 ,6755.9  ,61.3,85.5,108.4
XS GIS Cut Line= 4
     1852996.185      370534.971     1853017.444      370617.784
     1853094.353      370760.671      1853160.13      370819.085
#Sta/Elev= 26
       0 1271.23     9.5 1270.33      19 1269.89      38 1269.48    66.5 1268.56
    85.5 1267.67   114.1 1266.62   152.3 1265.06   171.4 1264.05     200 1261.97
   204.1 1261.94   209.6 1261.91   218.11261.937   219.1 1261.94   228.7  1262.7
   238.2 1266.08   247.8 1271.12   257.5 1276.85   267.3 1282.94   277.1 1289.37
   286.9 1295.94   296.6 1302.22   306.4 1308.17   316.2 1313.03     326 1314.67
   335.7 1315.16
#Mann= 3 , 0 , 0
       0     .08       0   204.1    .045       0   218.1     .08       0
#XS Ineff= 2 , 0
       0     130    1270               0
Permanent Ineff=
       F       F
Bank Sta=204.1,218.1
XS Rating Curve= 0 ,0
Exp/Cntr=0.3,0.1

Type RM Length L Ch R = 1 ,6670.4  ,54.4,54.5,60.9
XS GIS Cut Line= 6
     1852900.321      370510.659     1853026.222      370659.422
     1852970.714      370758.392     1852955.031      370791.172
     1852944.198      370822.208     1853051.872       370895.58
#Sta/Elev= 30
       0  1319.3    19.5 1306.32    48.7 1286.65    58.5 1280.98    68.2 1277.24
      78 1275.44   107.2 1271.35   126.7 1269.13   136.4 1268.22   155.9 1266.91
   185.1 1266.21   201.2 1265.37   207.6 1264.91   216.8 1263.82     226 1262.46
   235.2 1261.92   249.21261.965     272 1262.73   281.1 1262.57   326.6 1261.05
     353 1260.38   377.6 1259.97   414.9 1260.84   424.2 1261.36   433.5 1263.02
   442.8 1266.69   452.1 1271.56   470.7 1281.95   498.6 1297.92   507.9 1302.53
#Mann= 3 , 0 , 0
       0     .08       0   235.2    .045       0   249.2     .08       0
#XS Ineff= 2 , 0
       0                     275       0    1270
Permanent Ineff=
       F       F
Bank Sta=235.2,249.2
XS Rating Curve= 0 ,0
Exp/Cntr=0.3,0.1

Type RM Length L Ch R = 1 ,6615.9  ,187.7,153.4,112.1
XS GIS Cut Line= 6
     1852874.756      370532.534     1852971.092      370644.771
     1852922.522      370733.125     1852906.838      370765.904
     1852892.533      370804.842     1853043.623      370903.395
#Sta/Elev= 30
       0 1317.42    18.5 1306.11      37 1294.52    46.2 1288.98    55.5 1284.72
    64.7 1281.97   120.2 1271.13   157.1 1263.21   166.3 1259.57   175.5 1255.63
   179.8 1255.06   184.8 1254.39     194 1254.51     1981255.139   203.2 1255.95
   221.4 1260.62   230.5 1261.23   285.1 1259.68   326.6 1258.71   345.6  1259.2
   374.1 1259.43     412 1260.34   421.5  1260.7     431 1261.77   440.5 1264.74
     450 1269.58   459.5 1274.88     488  1291.5   497.5 1296.78     507 1301.22
#Mann= 3 , 0 , 0
       0     .08       0   179.8    .045       0     198     .08       0
#XS Ineff= 2 , 0
       0                     235       0    1270
Permanent Ineff=
       F       F
Bank Sta=179.8,198
XS Rating Curve= 0 ,0
Exp/Cntr=0.3,0.1

Type RM Length L Ch R = 1 ,6462.5  ,184.2,182.7,180.9
XS GIS Cut Line= 2
     1852737.696      370708.806     1853042.356         370908.
#Sta/Elev= 29
       0 1321.94     9.8 1315.78    19.7  1309.7    29.5 1303.79      59 1286.26
    68.9 1280.46    78.7 1274.61    88.5 1268.64   108.2 1255.18   114.9 1252.79
     118 1251.69   127.9 1251.48   131.91252.379   137.7 1253.68   147.6 1256.49
   157.4 1257.76   167.2 1258.13   196.8 1258.97   206.6 1259.12   226.3 1259.21
   255.8 1259.87   275.5 1260.46   285.3  1261.4   295.1 1264.46     305 1269.21
   314.8 1274.78   344.3 1292.08   354.2 1297.42     364 1301.66
#Mann= 3 , 0 , 0
       0      .1       0   114.9    .045       0   131.9     .08       0
Bank Sta=114.9,131.9
XS Rating Curve= 0 ,0
Exp/Cntr=0.3,0.1
